HEC-RAS study U101-00-00.prj: U101-00-00 2019 (Re-Study)

--- U101-00-00.g01 (geometry) --- (continued)

Type RM Length L Ch R = 1 ,91417.91,821.73,776.81,797.44
XS GIS Cut Line= 6
2973079.0192460313882690.57894862973086.0720534513880728.8440269
2973139.1398606913879209.87003082973157.7051122813877831.1972632
2972535.4973671913876568.61907972970697.9508454513874961.5957189
#Sta/Elev= 30
       0  164.16 2241.62  161.22 2466.51  162.03 2546.47  160.78 2576.45  162.04
 2646.42  160.25 2661.41  161.51 2826.33  159.89 2856.31  161.32 2921.28  160.29
 3376.05  160.52 3405.17  160.08 3423.66  156.41 3442.12   160.7 3481.64  160.97
 3506.62  157.96 3526.61  160.97 4071.14  159.49 4820.49   160.4 4925.34  162.01
 4995.22  160.65 5219.84  160.57 6148.26  160.75 6377.88  162.13  6432.8  160.43
 6462.75  161.54 7825.61  161.12 8464.61  163.71 8489.57  162.68 8709.22  162.83
#Mann= 3 ,-1 , 0
       0     .07       0 3376.05     .04       0 3442.12     .07       0
#XS Ineff= 5 ,-1
       0 2856.31  161.32 2856.31 3376.05  160.52 3462.52 4875.43  160.52
 4875.43 6307.99  161.15 6307.99 8709.22   161.5
Permanent Ineff=
       F       F       F       F       F
Bank Sta=3376.05,3442.12
XS Rating Curve= 0 ,0
Exp/Cntr=0.5,0.3

Type RM Length L Ch R = 1 ,90641.11,50.38,50.22,51.48
BEGIN DESCRIPTION:
Upstream Section - DRIVEWAY #1
END DESCRIPTION:
Node Name=AY
XS GIS Cut Line= 6
 2973885.230045113880380.42326322973898.78368261 13879974.145077
2973912.2058998613879295.30850822973912.8997961113879263.3410524
2973966.6326282813876579.52719442971392.3073963713873890.5522574
#Sta/Elev= 30
    2166  160.93 3222.24  160.07 3232.24  159.96 3249.04  155.71 3253.89  155.66
 3256.29  157.44 3275.27   160.5  3318.4  159.86 3333.38  157.89 3348.36  160.21
 4491.93  159.41 4676.69  160.83 4716.57  159.81 5130.32  159.74  5200.1  158.46
 5912.94  158.49 5942.85  158.59 5967.77  161.56 6017.74  158.55 6957.15  158.12
 7681.69  159.88 8041.46  159.46  8151.4  160.69  8656.1  160.39 9625.53  162.23
 9640.52  162.06 9650.51  160.13 9660.51  159.83  9675.5  161.88 9690.49  162.17
#Mann= 3 ,-1 , 0
    2166     .07       0 3222.24     .04       0 3275.27     .07       0
#XS Ineff= 4 ,-1
    2166 3245.36  159.65 3256.56 3293.43   160.7 4696.63 5967.77  160.65
 5967.77 9690.49  161.56
Permanent Ineff=
       F       F       T       T
#Block Obstruct= 2 , 0
       0                 9625.53       0  162.23
Bank Sta=3222.24,3275.27
XS Rating Curve= 0 ,0
Exp/Cntr=0.5,0.3

Type RM Length L Ch R = 2 ,90618.37,,,
BEGIN DESCRIPTION:
DRIVEWAY #1
END DESCRIPTION:
Node Name=DRIVEWAY #1
Bridge Culvert--1,0,-1,-1, 0
Deck Dist Width WeirC Skew NumUp NumDn MinLoCord MaxHiCord MaxSubmerge Is_Ogee
21,14,2.6,0, 10, 10, , , 0.98, 0, 0,0,,
 2697.44 2727.43 2757.42 2862.38 2887.37 2917.36 2997.33 3117.28 3246.66 3293.43
  160.69  161.05  160.82  160.49  160.48  160.19  160.11  160.34  160.71  160.88
       0       0       0       0       0       0       0       0       0       0
 2697.44 2727.43 2757.42 2862.38 2887.37 2917.36 2997.33 3117.28 3246.66 3293.43
  160.69  161.05  160.82  160.49  160.48  160.19  160.11  160.34  160.71  160.88
       0       0       0       0       0       0       0       0       0       0
BR Coef=-1 , 0 , 0 ,, 0 ,,,0.8,-1,,0,
WSPro=,,,, 1 ,,,, 0 ,,,, 0 ,,,,-1 ,-1 ,-1 , 0 , 0 , 0 , 0 , 0
Culvert=1,3,,23.8,0.013,0.5,1,1,3,155.61,3246.86,156.43,3246.86,Culvert #1  , 0 ,18.5
Culvert Bottom n=0.013
Culvert=1,3,,23.8,0.013,0.5,1,1,3,155.62,3250.96,156.04,3250.96,Culvert #2  , 0 ,18.5
Culvert Bottom n=0.013
Culvert=1,3,,23.8,0.013,0.5,1,1,3,155.79,3255.06,156.19,3255.06,Culvert #3  , 0 ,18.5
Culvert Bottom n=0.013
BC Design=,, 0 ,, 0 ,,,,,,
BC Use User HTab Curves=0
BC User HTab FreeFlow(D)= 0

Type RM Length L Ch R = 1 ,90590.89,811.68,751.27,788.88
BEGIN DESCRIPTION:
Downstream Section - DRIVEWAY #1
END DESCRIPTION:
XS GIS Cut Line= 6
2973934.9679934413882548.94832632973930.6484482713880523.7177968
2973948.8954590313879976.75301142973962.3176762813879297.9164426
2974016.7444046913876582.13512882971442.4191727813873893.1601918
#Sta/Elev= 30
       0  163.69   19.95  162.65 1935.44  161.53 1960.39   163.1 1975.35  161.81
 2139.66  161.24 3207.25  158.64 3232.24  159.53 3253.41  155.56 3269.74  160.12
 3303.42  160.47 3333.38  157.96 3358.35  160.51 3503.17  159.37 4566.83  159.39
 4696.63  160.82 5080.47  159.77 5175.18  158.46 5823.21  158.14 5932.88  159.25
 5942.85  158.04 5967.77  161.31 5987.76  159.52 6032.73  158.52 6892.19  157.93
 7042.09  159.73 7152.03  158.04 9630.53  162.38 9655.51  159.64 9690.49  162.12
#Mann= 3 ,-1 , 0
       0     .07       0 3232.24     .04       0 3269.74     .07       0
#XS Ineff= 4 ,-1
       0 3245.36     159 3256.56 4696.63     159 4696.63 5967.77   160.6
 5967.77 9690.49   161.5
Permanent Ineff=
       F       F       T       F
#Block Obstruct= 2 , 0
       0                 9630.53       0  162.38
Bank Sta=3232.24,3269.74
XS Rating Curve= 0 ,0
Exp/Cntr=0.5,0.3

Type RM Length L Ch R = 1 ,89839.63,55.03,47.77,47.63
Node Name=AX
XS GIS Cut Line= 6
2974685.0791871713880104.47260282974710.8585020313879362.3569305
2974715.2872989513879242.22331252974765.9981555313877899.3483736
2974836.8671082713876029.66805792972029.3051381113872679.4237741
#Sta/Elev= 30
 1739.67  160.15 2491.42  158.88 2504.68   158.6 2519.37  154.93 2543.53  159.65
  2577.9  159.81 2602.45  156.84 2632.42  159.83 2642.41  158.49 3346.79  158.61
 3956.24  160.46 4001.15  159.06 4415.26  159.67 4904.21   157.9 5128.72  159.04
 5408.12  157.29 5487.95  158.87 5507.91  157.54 5657.58  157.18 6596.55  157.54
 6681.48  159.11 6716.45  157.29 8474.89  158.87 8504.86  156.59 8539.83  158.19
 8559.81  156.48  8574.8  158.81 8689.69  157.34 8839.55  159.8210188.33  160.74
#Mann= 3 ,-1 , 0
 1739.67     .07       0 2491.42     .04       0 2543.53     .07       0
#XS Ineff= 3 ,-1
       0 2043.67   159.8 3956.24    4950   159.8    495010188.33  160.46
Permanent Ineff=
       F       T       F
Bank Sta=2491.42,2543.53
XS Rating Curve= 0 ,0
Exp/Cntr=0.3,0.1

Type RM Length L Ch R = 1 ,89791.85,57.85,47.12,47.08
XS GIS Cut Line= 6
2974671.7683571113881841.27782572974713.4293630313880660.5016439
2974758.5860968513879360.56329892974813.72575036 13877897.554742
2974884.5947031113876027.87442632972077.0327329513872677.6301425
#Sta/Elev= 30
       0  162.17 1420.72  161.63 1440.66  160.24 1595.15  159.67 2496.02  158.89
 2517.35  155.15  2539.8  159.42 2572.99  159.74 2597.54  156.92 2622.43  159.51
  2657.4  160.36 2677.38  158.94 3931.28  158.99 3966.22  160.13  5697.5  156.97
 6621.53  157.41 6646.51  158.85 6706.46  157.23  8464.9  158.93 8499.86   156.2
 8534.83  158.17 8554.81  156.51  8574.8  159.53 8724.66  157.32  9009.4  159.53
 9314.12  159.61  9339.1  160.87 9593.87  159.71  9993.5  161.8210188.33  160.75
#Mann= 3 ,-1 , 0
       0     .07       0 2496.02     .04       0  2539.8     .07       0
#XS Ineff= 3 ,-1
       0 2038.69   159.7 3966.22 4944.12   159.7 4944.1210188.33   160.3
Permanent Ineff=
       F       T       F
Bank Sta=2496.02,2539.8
XS Rating Curve= 0 ,0
Exp/Cntr=0.3,0.1

Type RM Length L Ch R = 1 ,89744.73,60.84,50.49,49.88
XS GIS Cut Line= 6
2974718.80435228 13881842.594096 2974760.465358213880661.8179143
2974805.6220920213879361.87956932974860.7617455313877898.8710123
2974931.6306982813876029.1906966 2972124.068728113872678.9464128
#Sta/Elev= 30
       0  162.15 1196.46  160.58 1226.36  162.02 1804.46   158.9 2477.25  158.33
 2510.38  157.45  2518.5  155.52 2536.38  159.15 2558.26  160.36 2597.54  157.18
 2627.43  159.98 3366.77  158.51 3826.37  158.65 3946.26  160.17 4884.25  158.15
  4904.2  159.45 5173.62  156.95 5213.54  158.65 6346.77  157.08 6671.49  158.71
 6906.28  157.24 8479.88  158.58 8494.87  156.31 8514.85  157.99 8554.81  156.49
  8569.8  158.11 8819.57  157.42  9334.1  160.69 9583.88  159.6710188.33   161.1
#Mann= 3 , 0 , 0
       0     .07       0 2477.25     .04       0 2536.38     .07       0
#XS Ineff= 3 ,-1
       0 2038.69   159.6 4026.09  4904.2  159.65  4904.210188.33  160.15
Permanent Ineff=
       F       T       F
Bank Sta=2477.25,2536.38
XS Rating Curve= 0 ,0
Exp/Cntr=0.5,0.3

Type RM Length L Ch R = 1 ,89694.23,169.1,151,150.5
BEGIN DESCRIPTION:
Upstream Section - KATY HOCKLEY RD
END DESCRIPTION:
XS GIS Cut Line= 6
2974768.6897511913881842.42382082974810.35075711 13880661.647639
2974855.50749095 13879361.7092942974910.6471444413877898.7007371
2974981.5160971913876029.02042142972173.9541270313872678.7761376
#Sta/Elev= 30
       0  162.31 1161.57  162.03 1186.49  160.49 1196.46  162.12 1630.03  159.13
 2282.89  158.01 2482.23  159.54 2520.22  155.22 2533.13  155.99 2535.74  159.53
 2572.99   159.8 2597.54     157 2672.39  159.48  3456.7  158.33  4629.8  159.98
 4849.32  158.04 4899.22  159.67 4939.13  158.08 5243.47  157.42 5353.24  158.99
  5373.2  157.59 5448.03  158.82 5792.29  156.95 8474.89  158.28 8494.87  156.09
 8549.82  156.48 8579.79  158.66 8799.59  157.09 9384.06  160.7210188.33  161.09
#Mann= 3 ,-1 , 0
       0     .07       0 2482.23     .04       0 2535.74     .07       0
#XS Ineff= 3 ,-1
       0  2511.4  159.34 2533.55    5250   158.8    525010188.33   160.1
Permanent Ineff=
       F       F       F
#Block Obstruct= 2 , 0
       0                10143.37       0  161.55
Bank Sta=2482.23,2535.74
XS Rating Curve= 0 ,0
Exp/Cntr=0.5,0.3

Type RM Length L Ch R = 2 ,89615.38,,,
BEGIN DESCRIPTION:
KATY HOCKLEY RD
END DESCRIPTION:
Node Name=KATY HOCKLEY RD
Bridge Culvert--1,0,-1,-1, 0
Deck Dist Width WeirC Skew NumUp NumDn MinLoCord MaxHiCord MaxSubmerge Is_Ogee
60,41.2,2.6,0, 52, 52, , , 0.98, 0, 0,0,,
       0   19.94  109.68  244.28  368.91  533.42  613.19  697.94  857.47 1036.94
 1076.82 1201.44  1246.3 1321.05 1585.18 1729.71 1809.44 1844.33 1864.26 1909.12
 1998.82 2063.61 2103.48  2158.3 2193.18 2213.12  2402.5 2417.45 2427.41 2513.64
 2513.74 2530.21 2538.21 2538.31 2677.38 2842.24  2887.2 3087.02 3136.98 3241.88
 3426.72 3636.54 3881.32 3911.29  4021.1    4071 4235.64 4664.72 5193.58 5318.31
 5817.24 5837.22
  162.04  162.12  162.16  161.98  161.82  161.81  161.87  161.72   161.4  161.33
  161.21  161.18  161.19   160.9  160.39   160.1  159.86  159.84  159.98  159.97
  159.82  159.52   159.6   159.6  159.52  159.36  159.34  159.37  159.45  159.71
  162.29  162.18  162.28  159.78  159.84  160.06  159.99  159.72   159.6  159.22
  159.32  159.43  159.71  159.61  159.24  159.35  159.35  159.12  159.03  158.75
  158.43   157.7
       0       0       0       0       0       0       0       0       0       0
       0       0       0       0       0       0       0       0       0       0
       0       0       0       0       0       0       0       0       0       0
       0       0       0       0       0       0       0       0       0       0
       0       0       0       0       0       0       0       0       0       0
       0       0
       0   19.94  109.68  244.28  368.91  533.42  613.19  697.94  857.47 1036.94
 1076.82 1201.44  1246.3 1321.05 1585.18 1729.71 1809.44 1844.33 1864.26 1909.12
 1998.82 2063.61 2103.48  2158.3 2193.18 2213.12  2402.5 2417.45 2427.41 2513.64
 2513.74 2530.21 2538.21 2538.31 2677.38 2842.24  2887.2 3087.02 3136.98 3241.88
 3426.72 3636.54 3881.32 3911.29  4021.1    4071 4235.64 4664.72 5193.58 5318.31
 5817.24 5837.22
  162.04  162.12  162.16  161.98  161.82  161.81  161.87  161.72   161.4  161.33
  161.21  161.18  161.19   160.9  160.39   160.1  159.86  159.84  159.98  159.97
  159.82  159.52   159.6   159.6  159.52  159.36  159.34  159.37  159.45  159.71
  162.29  162.18  162.28  159.78  159.84  160.06  159.99  159.72   159.6  159.22
  159.32  159.43  159.71  159.61  159.24  159.35  159.35  159.12  159.03  158.75
  158.43   157.7
       0       0       0       0       0       0       0       0       0       0
       0       0       0       0       0       0       0       0       0       0
       0       0       0       0       0       0       0       0       0       0
       0       0       0       0       0       0       0       0       0       0
       0       0       0       0       0       0       0       0       0       0
       0       0
BR Coef=-1 , 0 , 0 ,, 0 ,,,0.8,-1,,0,
WSPro=,,,, 1 ,,,, 0 ,,,, 0 ,,,,-1 ,-1 ,-1 , 0 , 0 , 0 , 0 , 0
Culvert=2,4,8,41.2,0.015,0.5,1,10,1,154.56,2518.4,154.41,2518.4,Culvert #1  , 0 ,60
Culvert Bottom n=0.015
Culvert=2,4,8,41.2,0.015,0.5,1,10,1,154.55,2527.55,154.42,2527.55,Culvert #2  , 0 ,60
Culvert Bottom n=0.015
BC Design=,, 0 ,, 0 ,,,,,,
BC Use User HTab Curves=0
BC User HTab FreeFlow(D)= 0

Type RM Length L Ch R = 1 ,89543.23,50.06,50.26,49.83
BEGIN DESCRIPTION:
Downstream Section - KATY HOCKLEY RD
END DESCRIPTION:
XS GIS Cut Line= 6
2974918.8938471113881850.11835922974960.5548530213880669.3421774
2975005.7115868613879369.40383242975060.8512403713877906.3952755
 2975131.720193113876036.71495982972324.15822294 13872686.470676
#Sta/Elev= 30
       0  161.69 1679.87  158.66 2422.43  159.77 2491.42  158.95    2521  154.88
 2538.62     160 2568.08  160.28 2602.45  157.38 2627.43  159.57 2687.37  159.67
 5144.25  157.76 5253.45  159.06 5537.84  156.73 5840.46  158.04 5887.18  156.17
 5897.17  157.94 5942.13  157.88 5957.12  156.04  5977.1  158.49  6546.6  157.03
 6676.48  158.85 6846.33  157.12 8484.88  157.93 8499.86  156.08 8514.85   157.7
 8554.81  156.29  8574.8   157.8 8954.45  156.73 9439.01   160.810188.33  160.93
#Mann= 5 ,-1 , 0
       0     .07       0 2422.43     .04       0 2538.62     .07       0
 5144.25      .1       0 5840.46     .07       0
#XS Ineff= 3 ,-1
       0  2513.4  158.93 2531.55 6027.05     158 6027.0510188.33  159.25
Permanent Ineff=
       F       F       T
Bank Sta=2422.43,2538.62
XS Rating Curve= 0 ,0
Exp/Cntr=0.5,0.3

Type RM Length L Ch R = 1 ,89492.98,53.22,51.02,51.04
XS GIS Cut Line= 6
2974968.40063787 13881858.5586312975010.0616437813880677.7824493
2975055.2183776113879377.84410432975110.3580311113877914.8355474
2975181.2269838613876045.1552316 2972373.665013713872694.9109479
#Sta/Elev= 30
       0  161.73 1839.35  158.27 2477.25  159.72 2499.43  158.93 2519.86  154.44
 2543.53  159.44 2563.17  160.26 2607.44  157.23 2637.42  159.79 5151.17  157.75
 5193.58  158.23 5213.54  155.49 5253.45  158.54    5849  158.01 5962.11  156.21
 5997.08  158.43 6032.05  155.67 6057.03  158.64 6601.55  157.24  6651.5  158.88
 6661.49  157.12 6681.48  158.63 6741.42  157.21 8479.88  158.29 8509.86  155.84
 8534.83  157.99 8564.81  156.31 8959.45  156.47 9528.93  160.5710188.33  160.89
#Mann= 5 ,-1 , 0
       0     .07       0 2477.25     .04       0 2563.17     .07       0
 5151.17      .1       0    5849     .07       0
#XS Ineff= 3 ,-1
       0 2382.82  158.93 2637.42 6057.03     158 6057.0310188.33   159.2
Permanent Ineff=
       F       F       T
Bank Sta=2477.25,2563.17
XS Rating Curve= 0 ,0
Exp/Cntr=0.3,0.1

Type RM Length L Ch R = 1 ,89441.95,46.28,43.68,43.7
XS GIS Cut Line= 6
2975019.3637905313881860.69412542975061.0247964413880679.9179437
2975106.1815302813879379.97959872975161.3211837713877916.9710418
2975232.19013652 13876047.2907262972424.6281663613872697.0464423
#Sta/Elev= 30
       0  161.77 1091.77  161.73 1799.48  158.21 2486.83  159.77 2509.06  158.34
 2516.31  154.14 2563.17  160.11 2607.44  157.31 2617.44  159.25 5151.74  157.93
 5193.58  158.93 5208.55  155.88  5278.4  158.83 5458.01  157.46 5552.81  159.12
  5602.7  157.07 5767.35  156.63 5848.93  158.39 6042.04  155.81    6087  158.28
 6106.98     156 6131.96  158.51 8484.88  158.07 8509.86  155.88 8604.77  158.12
 9024.39  157.07 9039.37  160.01 9079.34   156.8 9359.08  160.2410188.33  160.82
#Mann= 5 ,-1 , 0
       0     .07       0 2486.83     .04       0 2563.17     .07       0
 5151.74      .1       0 5848.93     .07       0
#XS Ineff= 2 ,-1
       0 2088.53  158.85 5552.8110188.33  159.12
Permanent Ineff=
       F       T
Bank Sta=2486.83,2563.17
XS Rating Curve= 0 ,0
Exp/Cntr=0.3,0.1

Type RM Length L Ch R = 1 ,89398.27,703.01,673.08,573.9
Node Name=AW
XS GIS Cut Line= 6
2975116.2917671813880346.75257492975149.8566397713879380.5120779
2975154.2854366913879260.37845992975204.99629328 13877917.503521
2975275.8652460313876047.82320532972468.3032758513872697.5789215
#Sta/Elev= 30
 1515.41  159.71 2337.71   158.2 2491.42  159.75 2508.22  158.18 2516.24  154.34
 2563.17  160.02 2607.44  157.31 2622.43  159.57 5150.93  157.82 5193.58  158.84
 5213.54  155.31 5223.52  157.65 5303.35  158.69 5847.11  158.51 6101.99  155.35
 6141.95  158.57 6171.93  156.01  6196.9  158.43 6681.48  158.81 6856.32  157.11
 8479.88  157.96 8504.86  155.46 8524.84  157.73 8564.81  156.09 9029.38  156.42
 9054.36     160 9079.34  156.64 9154.27  156.27 9374.07  160.5110188.33  160.79
#Mann= 5 ,-1 , 0
 1515.41     .07       0 2491.42     .04       0 2563.17     .07       0
 5150.93      .1       0 5847.11     .07       0
#XS Ineff= 2 ,-1
 1515.41 2163.28   158.8  5557.810188.33   159.1
Permanent Ineff=
       F       T
Bank Sta=2491.42,2563.17
XS Rating Curve= 0 ,0
Exp/Cntr=0.3,0.1

Type RM Length L Ch R = 1 ,88725.2 ,1153.65,1141.28,881.85
XS GIS Cut Line= 6
 2975775.132620213881945.38358862975759.1536495213880363.8903605
2975820.95995636 13879405.1698372975825.8900646113879302.2901215
2975722.9115960313876050.02005132972557.7673357713872238.2343678
#Sta/Elev= 30
       0  159.89  2537.3  158.86  2566.3  157.21 2580.56  152.92 2602.27  158.11
 2625.66  159.25 2665.27  156.22 2685.27  158.58 3105.13  161.08    3490   157.6
 5220.08     157 5244.38  154.82 5264.37  157.81 5906.05  158.33 6239.11  155.83
 6689.06  158.05 6859.05   156.1 6889.04  158.18 6924.04  155.98 6964.04  158.22
 7513.98  156.98 8403.91  158.98 8423.91   157.1  8618.9  155.37  8633.9  157.18
 8963.89  158.17 9033.89  156.08 9283.88  156.32 9713.87  159.9310853.84  161.23
#Mann= 6 ,-1 , 0
       0     .07       0  2537.3     .04       0 2625.66     .05       0
 2685.27     .07       0 5220.08      .1       0 5906.05     .07       0
#XS Ineff= 3 ,-1
       0  2537.3   158.7 3105.13 6964.04   157.9 6964.0410853.84  158.22
Permanent Ineff=
       F       T       T
Bank Sta=2537.3,2625.66
XS Rating Curve= 0 ,0
Exp/Cntr=0.3,0.1

Type RM Length L Ch R = 1 ,87583.91,343.88,344.22,208
XS GIS Cut Line= 6
2976647.3700489413881994.38545912976923.0617547813879829.2972696
2976966.2700016913879342.95014522976984.2624197813879058.1912003
 2976227.263605713876068.90059092972736.8211115313871987.3086885
#Sta/Elev= 30
       0  160.25 1992.78  157.42 2571.19  158.76 2606.26  152.98 2630.97  157.93
  2650.9  158.56 2690.51  155.58 2705.27   157.7 3970.72  156.81 4010.71  153.31
 4040.69  157.62 5338.36  155.57 5365.08   154.3 5385.07  157.28 5400.06  155.25
 5425.05  157.24 5440.04  154.15 5619.96  154.24 5649.94  159.35  5734.9  156.59
 6042.96  157.93 7728.36  155.35 7748.34  157.65  7793.3  155.18 7873.24  158.55
 8148.01  158.77 8897.41  155.05 9047.29  159.01 9132.23  156.3111410.41  160.48
#Mann= 5 ,-1 , 0
       0     .07       0 2571.19     .04       0  2650.9     .07       0
 5338.36      .1       0 6042.96     .07       0
#XS Ineff= 3 ,-1
       0 2571.19  157.73 5649.94 7873.24  157.66 7873.2411410.41  158.55
Permanent Ineff=
       F       F       F
#Block Obstruct= 1 ,-1
 5425.05 5649.94  157.24
Bank Sta=2571.19,2650.9
XS Rating Curve= 0 ,0
Exp/Cntr=0.3,0.1

Type RM Length L Ch R = 1 ,87239.7 ,487.27,270.89,76.99
XS GIS Cut Line= 6
2977039.3869814413881984.58528182977185.8801267713880285.7100707
 2977302.729958713879498.81991222977268.0699230313878952.5398368
2976338.0950769513876071.20636062972919.1130697713871674.8086573
#Sta/Elev= 30
       0  160.36 2544.75  157.53 2564.32   157.1 2576.81  151.96 2608.37  157.89
  2662.2   155.3 3953.22  156.75  3988.2   152.3 4018.17  157.09 5359.24  155.78
 5427.11  155.09 5447.09  158.39 5472.07  158.13 5497.06  154.18 5636.95  153.91
 5676.92   158.8 5771.85  156.48  6076.3  157.87 7081.52  155.82 7421.48  158.02
 8026.42  154.91 8051.42  157.87 8096.41   155.4  8156.4  158.49 8486.34   158.2
 8666.31  155.29  8696.3  157.41  8721.3  155.05 8751.29  157.5511645.73  160.09
#Mann= 5 ,-1 , 0
       0     .07       0 2544.75     .04       0 2608.37     .07       0
 5359.24      .1       0  6076.3     .07       0
#XS Ineff= 3 ,-1
       0 2544.75  157.53 5676.92  8156.4  157.53  8156.411645.73  158.49
Permanent Ineff=
       F       F       F
#Block Obstruct= 1 ,-1
 5462.08  5706.9  157.64
Bank Sta=2544.75,2608.37
XS Rating Curve= 0 ,0
Exp/Cntr=0.5,0.3

Type RM Length L Ch R = 1 ,86968.8 ,18.97,73.17,24.85
BEGIN DESCRIPTION:
Upstream Section - FREEMAN (FM 529)
END DESCRIPTION:
Node Name=AV
XS GIS Cut Line= 6
2977823.4060548313880688.51010952977634.1052801913879412.8561734
2977437.8100691113879403.10848942976473.8103566913876105.4940217
2975130.0240022813874034.87939652973199.9045029413871324.1220228
#Sta/Elev= 30
 1199.65  158.59 1584.53  158.45 1929.43  155.45 2434.29  157.11 2464.28  154.52
 2508.11  157.52 2532.89  155.37  2545.4  151.32 2613.26   157.6 2730.75   157.7
 2750.73  155.28 4059.07  156.49 4079.04  152.62 4099.02  152.75    4114  157.22
 5442.65  157.13  5467.3  154.46 5527.22  157.23 5746.95  155.82 5916.73  158.42
 6036.58  156.32 6156.15  157.43 8520.03  156.81 8540.02  154.04    8570  157.65
 8624.96  157.55 8644.95  154.77 8654.94  156.82 8744.88  157.0811917.62   159.8
#Mann= 5 ,-1 , 0
 1199.65     .07       0 2508.11     .04       0 2613.26     .07       0
 5442.65      .1       0 6156.15     .07       0
#XS Ineff= 4 ,-1
 1199.65 2508.11   157.2 2508.11 2524.03  155.45 2577.69    8570  156.69
    857011917.62  157.65
Permanent Ineff=
       F       F       F       F
Bank Sta=2508.11,2613.26
XS Rating Curve= 0 ,0
Exp/Cntr=0.5,0.3

Type RM Length L Ch R = 3 ,86946.31,,,
BEGIN DESCRIPTION:
FREEMAN (FM 529)
END DESCRIPTION:
Node Name=FREEMAN (FM 529)
Bridge Culvert--1,0,-1,-1, 0
Deck Dist Width WeirC Skew NumUp NumDn MinLoCord MaxHiCord MaxSubmerge Is_Ogee
7,35,2.6,0, 36, 35, , , 0.98, 0, 0,0,,
 1929.43 2004.41 2059.39 2139.37 2219.35  2250.5 2274.33 2319.32 2339.31 2349.31
 2359.31  2384.3 2404.29 2414.29 2429.29 2439.28 2444.28 2454.28 2474.27  2517.7
 2577.69  2618.1 2676.14 2710.78 2725.76 2740.74 2780.69 2790.68 2825.63  2907.3
 2955.47 2985.43 3020.39 3070.32  3090.3 3125.25
  155.45  155.76  155.79  155.68  155.74  155.71  157.62  158.41  158.45  158.47
  158.49  158.51  158.53  158.54  158.56  158.56  158.57  158.58  158.59  158.63
  158.69  158.72  158.77  158.81  158.82  158.84  158.19   158.2  158.24   156.9
  156.91  156.78  156.89  156.71  156.88   156.7
       0       0       0       0       0       0       0       0       0       0
       0       0       0       0       0       0       0       0       0  156.38
  156.44       0       0       0       0       0       0       0       0       0
       0       0       0       0       0       0
 1789.47 2004.41 2059.39 2219.35  2250.5 2274.33 2319.32 2339.31 2349.31 2359.31
  2384.3 2404.29 2414.29 2429.29 2439.28 2444.28 2454.28 2474.27  2517.7 2577.69
  2618.1 2676.14 2710.78 2725.76 2740.74 2780.69 2790.68 2825.63  2907.3 2955.47
 2985.43 3020.39 3070.32  3090.3 3125.25
  155.47  155.76  155.79  155.74  155.71  157.62  158.41  158.45  158.47  158.49
  158.51  158.53  158.54  158.56  158.56  158.57  158.58  158.59  158.63  158.69
  158.72  158.77  158.81  158.82  158.84  158.19   158.2  158.24   156.9  156.91
  156.78  156.89  156.71  156.88   156.7
       0       0       0       0       0       0       0       0       0       0
       0       0       0       0       0       0       0       0  156.35  156.41
       0       0       0       0       0       0       0       0       0       0
       0       0       0       0       0
Pier Skew, UpSta & Num, DnSta & Num=  ,2538, 2 ,2538, 2 , 0 , 0 , 0 ,,
     2.2     2.2
     150   157.5
     2.2     2.2
     150   157.5
Pier Skew, UpSta & Num, DnSta & Num=  ,2557.5, 2 ,2557.5, 2 , 0 , 0 , 0 ,,
     2.2     2.2
     150   157.5
     2.2     2.2
     150   157.5
Abutment Skew #Up #Dn= , 2 , 2
  2517.5  2518.8
  156.38  154.77
  2517.5  2518.8
  156.35  154.74
Abutment Skew #Up #Dn= , 3 , 3
  2576.5 2577.89 2578.89
  154.57  156.44  156.44
  2576.5 2577.89 2578.89
  154.54  156.41  156.41
BR Coef=-1 , 1 , 1 ,0.9, 0 ,,,0.8,-1,1.2,0,
WSPro=,,,, 1 ,,,, 0 ,,,, 0 ,,,,-1 ,-1 ,-1 , 0 , 0 , 0 , 0 , 0
BC Design=,, 0 ,, 0 ,,,,,,
BC Use User HTab Curves=0
BC User HTab FreeFlow(D)= 0

Type RM Length L Ch R = 1 ,86895.63,654.33,248.52,270.24
BEGIN DESCRIPTION:
Downstream Section - FREEMAN (FM 529)
END DESCRIPTION:
XS GIS Cut Line= 6
2978004.4277022813881803.49345242977639.0330918613879341.1840726
2977442.7378807813879331.43638872976478.7381683613876033.8219209
2975134.9518139413873963.20729582973204.83231461 13871252.449922
#Sta/Elev= 30
       0  159.17 1514.56  158.32 1789.47  155.47 2334.31  155.74 2364.31  157.26
  2389.3  154.59 2424.29  157.61 2479.27  157.48 2536.38  154.88 2555.22  151.59
 2598.75  157.53 2705.78  155.53 3984.16  156.45 4004.14  152.44 4024.11     153
 4044.09  157.56 5367.14  156.65 5397.39  155.12 5412.37  157.99 5477.29  155.97
 5652.07  155.88 5896.76  158.32 6281.38  156.28 8475.06  156.99 8495.04  153.74
 8515.03  156.67    8580  157.68 8619.97  154.15 8649.95  157.2311917.63  158.46
#Mann= 5 ,-1 , 0
       0     .07       0 2479.27     .04       0 2598.75     .07       0
 5367.14      .1       0 6281.38     .07       0
#XS Ineff= 4 ,-1
       0 2444.28  157.15 2444.28 2517.54  155.45 2577.69    8580   156.6
    858011917.63  157.68
Permanent Ineff=
       F       F       F       F
Bank Sta=2479.27,2598.75
XS Rating Curve= 0 ,0
Exp/Cntr=0.5,0.3

Type RM Length L Ch R = 1 ,86647.11,1103.1,903.23,403.25
Node Name=AU
XS GIS Cut Line= 5
2979122.98202364 13881158.1997382977961.6515411113879302.9223381
 2977644.930061713879130.38003232976790.7221244413876080.6233365
2973574.3348564513871310.0452793
#Sta/Elev= 30
  659.63  158.46 2643.51  157.44  2673.5  154.55 2733.46  157.49 2778.44  154.45
 2813.42  157.35 2991.68  157.49 3090.49  156.28 3108.11  151.07 3130.08  154.31
 3134.96  157.29 4273.12  156.07 4303.09  152.47 4348.05  156.59 5663.73  156.49
 5691.86  155.42 5701.85  158.14 6046.55  156.43 6116.49   158.7 6171.44  156.45
  6216.4  158.18 6365.63  156.63 8210.81  157.31 8880.68  155.15 8905.68  157.36
  9290.6  156.85 9350.59  153.95 9370.59  156.41 9430.57  156.8112130.05  159.65
#Mann= 5 ,-1 , 0
  659.63     .07       0 2991.68     .04       0 3134.96     .07       0
 5663.73      .1       0 6365.63     .07       0
#XS Ineff= 3 ,-1
  659.63 2991.69  157.05 3149.78 8905.68   156.6 8905.6812130.05  157.36
Permanent Ineff=
       F       F       F
Bank Sta=2991.68,3134.96
XS Rating Curve= 0 ,0
Exp/Cntr=0.3,0.1

Type RM Length L Ch R = 1 ,85743.88,1006.48,1004.18,870.6
XS GIS Cut Line= 6
2980435.73583178 13880635.6988722978931.5469110313878956.1428479
2978232.2599237713878428.74003132978001.9831533613878260.1773764
2976934.1598296913876083.60758252973824.02595811 13871319.650575
#Sta/Elev= 30
       0  156.67 1494.77  157.69 1519.77  154.87 1589.76  158.04 1649.75  154.78
 1674.74  157.72 2777.19  155.85    3031  158.05 3054.93  156.77 3078.42  149.19
 3097.04  155.24 3125.55  157.82 3580.87  155.69 3610.86  152.26 3675.84  156.24
 5055.51  156.54  5090.5  154.36 5435.42  156.59  6025.3  156.59 7800.09  157.16
 8195.04  156.29 8260.03  153.68 8290.03   156.9  9019.9  157.06  9044.9   154.9
 9089.89   157.7 9129.88  154.85 9179.87  157.16 9979.73  158.9511529.46   159.5
#Mann= 5 ,-1 , 0
       0     .07       0    3031     .05       0 3125.55     .07       0
 5435.42      .1       0  6025.3     .07       0
#XS Ineff= 4 ,-1
       0 1674.74   156.8 3675.84 8290.03     156 8290.03 9399.83   156.9
 9399.8311529.46  157.37
Permanent Ineff=
       F       F       F       F
#Block Obstruct= 2 , 0
       0  284.96  157.86               0
Bank Sta=3031,3125.55
XS Rating Curve= 0 ,0
Exp/Cntr=0.3,0.1

Type RM Length L Ch R = 1 ,84739.7 ,896.03,1124.69,1190.05
Node Name=AT
XS GIS Cut Line= 6
2980341.7917939413878781.54805282978935.5600263613877716.2900127
2978828.5500697813877635.32987282978648.9178831113877489.3432881
2977744.2605716913876100.46155142974137.4374047813871342.9756596
#Sta/Elev= 30
       0   160.3   34.98  156.04   74.96  154.41   94.95  156.99  134.94  154.01
  179.91  156.66 1304.38  154.29 1764.16  155.19 1793.98  157.48 1828.78  155.09
 1848.08  148.51 1851.73  151.78  1873.5  156.86  2948.6  157.07  3013.5  153.42
 3088.39   155.9 3937.22  157.01  3962.2  155.09 6300.34  156.57 6325.32  152.93
  6345.3  157.04 6365.28  157.18 6385.27  155.17    7989  155.44 8008.98  157.58
 8068.93  154.96 8273.77  158.06 8473.61  155.68 8603.51  157.99 9757.61  159.35
#Mann= 3 ,-1 , 0
       0     .07       0 1793.98     .05       0  1873.5     .07       0
#XS Ineff= 2 ,-1
       0  179.91  156.66 6365.28 9757.61  157.18
Permanent Ineff=
       F       F
Bank Sta=1793.98,1873.5
XS Rating Curve= 0 ,0
Exp/Cntr=0.5,0.3

Type RM Length L Ch R = 1 ,83615.02,35.28,40.69,36
BEGIN DESCRIPTION:
Upstream Section - 72" CULVERT
END DESCRIPTION:
XS GIS Cut Line= 6
2980418.06001411 13878367.1207322979610.0124176113876863.6322692
2979477.0851900313876677.05160562979004.1806240213875780.7279389
2977751.8652152713874128.68695172975212.4352547813871402.9479806
#Sta/Elev= 30
       0  158.72   19.96  156.69  209.62  157.06  244.55  154.23  309.43  156.44
  339.38   153.7  359.34  157.06 1725.74   155.2 1763.48   154.5 1781.78  147.75
 1793.46  153.14 1819.01  155.27 2635.13  155.12 2665.09   156.9 3708.92  154.03
 3923.72  155.83  3948.7  153.63 4303.36  153.97  4363.3  156.45 4383.29  153.38
 4563.12  153.45 4593.09  156.98 4732.96  157.17 4997.71  155.48 5017.69  151.74
 5037.67  155.27 5087.61  153.35 5102.59  155.85 7774.32  155.34 8748.15  157.73
#Mann= 3 ,-1 , 0
       0     .07       0 1725.74     .05       0 1819.01     .07       0
#XS Ineff= 4 ,-1
       0  359.34  157.06  359.34 1777.23  154.54 1786.73 4732.96  153.95
 4732.96 8748.15  155.85
Permanent Ineff=
       F       F       F       F
#Block Obstruct= 1 ,-1
  4363.3 4593.09  156.45
Bank Sta=1725.74,1819.01
XS Rating Curve= 0 ,0
Exp/Cntr=0.5,0.3

Type RM Length L Ch R = 2 ,83589.01,,,
BEGIN DESCRIPTION:
72" CULVERT
END DESCRIPTION:
Node Name=72" CULVERT
Bridge Culvert--1,0,-1,-1, 0
Deck Dist Width WeirC Skew NumUp NumDn MinLoCord MaxHiCord MaxSubmerge Is_Ogee
4,30,2.6,0, 12, 14, , , 0.98, 0, 1,1,,
 1725.74 1730.46  1739.9 1754.05  1768.2 1772.92 1777.64 1782.35 1790.91 1795.19
 1804.36 1823.89
  154.75  155.08  154.76  154.68  154.81  154.84  154.86  154.89  154.94  154.97
  155.02  154.73
       0       0       0       0       0       0       0       0       0       0
       0       0
 1711.59 1725.74 1730.46  1739.9 1754.05  1768.2 1772.92 1777.64 1782.35 1790.91
 1795.19 1804.36 1823.89 1828.78
  155.23  154.75  155.08  154.76  154.78  154.86  154.89  154.91  154.94  154.99
  155.02     155  155.89  155.78
       0       0       0       0       0       0       0       0       0       0
       0       0       0       0
BR Coef=-1 , 0 , 0 ,, 0 ,,,0.8,-1,,0,
WSPro=,,,, 1 ,,,, 0 ,,,, 0 ,,,,-1 ,-1 ,-1 , 0 , 0 , 0 , 0 , 0
Culvert=1,6,,32,0.013,0.5,1,1,3,147.74,1781.98,148.06,1772.68,Culvert #1  , 0 ,3
Culvert Bottom n=0.013
BC Design=,, 0 ,, 0 ,,,,,,
BC Use User HTab Curves=0
BC User HTab FreeFlow(D)= 0

Type RM Length L Ch R = 1 ,83574.32,146.46,60.21,80.66
BEGIN DESCRIPTION:
Downstream Section - 72" CULVERT
END DESCRIPTION:
XS GIS Cut Line= 6
2980441.1941541913878335.99185732979633.1465576913876832.5033944
2979500.2193301213876645.92273082979027.3147641113875749.5990642
2977774.9993553613874097.55807692975235.5693948613871371.8191058
#Sta/Elev= 30
       0  160.22   79.85  156.25  234.57  156.84  289.47  154.45  344.37   156.8
  369.32  154.09  409.25  156.76  673.77  154.93 1706.87  155.95 1761.16  154.49
 1772.48  148.37 1786.01  153.18 1828.78  155.78 3798.84  153.96 3933.71  155.49
 3973.67  153.92 4273.39  154.71 4313.35     157 4353.31  153.29 4563.12  153.37
 4598.08  156.99 4952.75   155.3 4977.73  151.93 4992.72   154.9 5062.64  156.19
 5112.58  153.58 5142.54  155.37 7389.79  156.62 7609.52  155.23 8748.15  158.39
#Mann= 3 ,-1 , 0
       0     .07       0 1706.87     .05       0 1828.78     .07       0
#XS Ineff= 4 ,-1
       0  409.25  156.76  409.25 1768.68   154.5 1776.68 4588.09  153.85
 4588.09 8748.15  155.85
Permanent Ineff=
       F       F       F       F
#Block Obstruct= 1 ,-1
 4313.35 4598.08   156.5
Bank Sta=1706.87,1828.78
XS Rating Curve= 0 ,0
Exp/Cntr=0.5,0.3

Type RM Length L Ch R = 1 ,83514.11,728.91,514.5,287.83
Node Name=AS
XS GIS Cut Line= 5
2980841.8117912713878396.31391512979683.1900927713876782.4798724
2979631.1800261913876722.56004482979092.8448167713875711.5131824
2975767.9052724413871380.5697445
#Sta/Elev= 30
       0  160.41   29.95  156.37  765.41  155.42  889.81  153.77  918.46  155.88
  968.38  152.83 1018.29  155.64 2016.43  154.69 2045.93  147.98 2061.06  153.11
 2085.94  155.35 3411.28  156.12 4335.44     153 4365.41  155.59 4470.32  153.37
 4555.24   156.9 4585.21  154.06 4695.11  153.54 4715.09   156.9 4859.96  153.19
 4879.94  156.83 5014.82  155.18  5034.8  158.73 5094.74  154.68 5164.68  155.03
 5194.65  151.63 5214.63  155.11 5444.42  156.23  5469.4  154.14 8671.43  156.86
#Mann= 5 ,-1 , 0
       0     .07       0  765.41     .12       0  889.81     .07       0
 2016.43     .04       0 2085.94     .07       0
#XS Ineff= 3 ,-1
       0  703.82   156.5 4558.88 7402.62     154 7402.62 8671.43  156.09
Permanent Ineff=
       F       F       F
Bank Sta=2016.43,2085.94
XS Rating Curve= 0 ,0
Exp/Cntr=0.3,0.1

Type RM Length L Ch R = 1 ,82999.61,941.86,999.25,975.59
XS GIS Cut Line= 6
2982887.9212161213878630.76390552981439.91033261 13877307.284269
2979898.1000960313876335.23011082979630.9444623613876136.0625301
2979193.6139721913875716.01678232976401.7232305313871414.4217109
#Sta/Elev= 30
       0  159.01   19.97  159.62   64.89  155.08 1232.19  155.37 2758.65  154.32
  3226.5  154.53  3246.5  152.41 3261.49   154.7 3286.49  154.79 3301.49  152.24
 3316.48  155.07 3656.42  154.18 3686.42  156.48 3701.42   153.5 3714.94  154.21
 3734.97  146.68 3741.01  150.93 3777.73  155.02 6021.35  154.68 6116.32  152.21
 6381.22  156.75 6506.17  153.03 6601.13   155.4 6651.11  153.34 6666.11  155.55
 7320.86  155.53 7345.85  154.08 7375.84  156.24 7420.82  153.86 9854.87  156.79
#Mann= 5 ,-1 , 0
       0     .07       0 1232.19     .12       0 2758.65     .07       0
 3714.94     .05       0 3777.73     .07       0
#XS Ineff= 4 ,-1
       0 1337.76   155.5 1337.76 3289.92     154  6036.5 7375.84     154
 7375.84 9854.87   155.5
Permanent Ineff=
       F       F       F       F
Bank Sta=3714.94,3777.73
XS Rating Curve= 0 ,0
Exp/Cntr=0.3,0.1

Type RM Length L Ch R = 1 ,82000.36,296.69,811.6,783.78
XS GIS Cut Line= 6
2982950.5726656213877581.35688362980238.6000711913875411.6801206
2980125.74990319 13875370.1700332979727.5079175213875135.9930079
2978781.8123023713874307.47465192977008.9976065313871495.0058673
#Sta/Elev= 30
       0  153.83   17.92  154.46 1109.82  153.17 1159.81  157.33 1219.77  153.24
 1609.48   156.2 2054.14  154.34 2079.12  150.91 2707.11  152.96 2823.57  154.29
 2858.55  148.42 2913.51  154.46 3083.38  156.89 3218.28  155.29 3268.25  151.31
 3487.52  153.38  3524.7  146.04 3554.86  152.35 3583.72  153.11 4135.15  153.49
 4190.03  156.41 4254.89  152.33 5232.79  155.31  5467.6  154.56  5482.6  150.76
  5497.6  154.49  5532.6  153.41 5552.59  156.59 6792.46  153.92 8637.21  155.84
#Mann= 5 ,-1 , 0
       0     .07       0   17.92     .12       0 2707.11     .07       0
 3487.52     .06       0 3583.72     .07       0
#XS Ineff= 4 ,-1
       0  544.91  155.25  544.91 3312.21  151.73 4927.37  6412.5  152.82
  6412.5 8637.21  154.91
Permanent Ineff=
       F       F       F       F
Bank Sta=3487.52,3583.72
XS Rating Curve= 0 ,0
Exp/Cntr=0.3,0.1

Type RM Length L Ch R = 1 ,81188.76,114.39,117.31,497.26
XS GIS Cut Line= 6
2982958.4286210213877322.11396382980319.5300274513875099.5101413
2980336.0398369413874641.99005892980264.08000711  13874579.27004
2979394.0764977813874161.27350072977807.8109695313871515.4766269
#Sta/Elev= 30
       0  153.89   16.68  154.24  617.21  153.18  691.88  156.58  721.74  153.02
 1375.77  154.59 1565.72  154.11 1590.71  150.82 1660.69  152.89 1675.69  150.71
 1700.68  153.94 2540.43  152.65 2703.53  155.89 2800.35  152.68 3375.18  153.04
 3385.18  150.56 3405.18  152.87 3674.09  155.12 3838.31  153.22 3927.07  152.16
 3945.07  145.51 3967.25  146.18 3979.57     152    3992  153.23 4859.18  154.83
 4898.98  149.84 4933.81  154.07 4968.63  154.29 7388.51   153.7 8053.48  156.19
#Mann= 5 ,-1 , 0
       0     .07       0   16.68     .12       0 2703.53     .07       0
 3838.31     .06       0    3992     .07       0
#XS Ineff= 3 ,-1
       0  691.88     155  691.88 3376.18  151.73 4245.94 8053.48  152.82
Permanent Ineff=
       F       F       F
Bank Sta=3838.31,3992
XS Rating Curve= 0 ,0
Exp/Cntr=0.5,0.3

Type RM Length L Ch R = 1 ,81071.45,133.22,130.39,145.01
BEGIN DESCRIPTION:
Upstream Section - KATY-HOCKLEY CUTOFF RD
END DESCRIPTION:
XS GIS Cut Line= 6
2982900.7476340213877138.41649652980342.8974347713874977.7735081
2980357.4243086113874509.49951032980371.5584666913874053.8770619
2979687.8754508613872777.29660982977875.4364904513871431.2973334
#Sta/Elev= 30
       0  153.84 1109.43  155.09  1354.3  153.27 1374.29  151.32 1424.27  154.67
 1594.18  152.42 2411.05  155.02 2443.75  152.36  2728.6  154.12 3248.34  151.02
 3288.32  153.46 3308.31  150.54  3323.3  152.56 3467.91  154.03 3672.26  152.66
  3786.9  150.05 3796.07  148.79 3800.96  145.43 3896.08  151.55 4079.41  152.83
 4104.18  147.63 4119.04  152.76 4143.82   150.2 4173.54  153.49 4193.36  150.42
 4342.55  149.07 4407.46  153.61  4612.2  154.12 4662.13  151.96 7978.34  154.74
#Mann= 4 ,-1 , 0
       0     .12       0 2411.05     .07       0 3672.26     .06       0
 3896.08     .07       0
#XS Ineff= 4 ,-1
       0 2393.77   154.9 2393.77  3784.1   152.2 3843.79 6914.49   152.2
 6914.49 7978.34   154.9
Permanent Ineff=
       F       F       F       F
#Block Obstruct= 1 ,-1
 4173.54 4422.44   151.5
Bank Sta=3672.26,3896.08
XS Rating Curve= 0 ,0
Exp/Cntr=0.5,0.3

Type RM Length L Ch R = 3 ,80995.45,,,
BEGIN DESCRIPTION:
KATY-HOCKLEY CUTOFF RD
END DESCRIPTION:
Node Name=KATY-HOCKLEY CUT
Bridge Culvert--1,0,-1,-1, 0
Deck Dist Width WeirC Skew NumUp NumDn MinLoCord MaxHiCord MaxSubmerge Is_Ogee
54.5,40.5,2.6,0, 29, 29, , , 0.98, 0, 0,0,,
  3328.3 3343.29  3408.1 3477.88 3547.66  3597.5 3637.37 3662.29 3705.99  3784.1
 3811.82 3843.79 3861.39 3916.01 3935.72 3955.54 3965.45 3985.26 4010.04 4019.95
 4059.59 4084.36 4089.32 4114.09    4124 4168.59 4267.68 4282.62 4292.61
  152.32  153.08  153.12  153.58  153.88  153.81  154.13  154.52  156.19  158.57
  158.87   158.9  158.76  156.39  155.83  155.29  155.29  154.76  154.61  154.34
   154.1   153.7  153.76  153.34  153.46  153.11  153.51  153.31  152.47
       0       0       0       0       0       0       0       0       0  154.27
  154.57   154.6       0       0       0       0       0       0       0       0
       0       0       0       0       0       0       0       0       0
  3328.3 3343.29  3408.1 3477.88 3547.66  3597.5 3637.37 3662.29 3705.99  3784.1
 3811.82 3843.79 3861.39 3916.01 3935.72 3955.54 3965.45 3985.26 4010.04 4019.95
 4059.59 4084.36 4089.32 4114.09    4124 4168.59 4267.68 4282.62 4292.61
  152.32  153.08  153.12  153.58  153.88  153.81  154.13  154.52  156.19  158.57
  158.87   158.9  158.76  156.39  155.83  155.29  155.29  154.76  154.61  154.34
   154.1   153.7  153.76  153.34  153.46  153.11  153.51  153.31  152.47
       0       0       0       0       0       0       0       0       0  154.22
  154.52  154.55       0       0       0       0       0       0       0       0
       0       0       0       0       0       0       0       0       0
Abutment Skew #Up #Dn= , 3 , 3
  3781.9  3783.9  3785.3
  154.27  154.27  149.05
  3781.9  3783.9  3785.3
  154.22  154.22     149
Abutment Skew #Up #Dn= , 3 , 3
  3841.3 3843.99 3845.99
  152.21   154.6   154.6
  3841.3 3843.99 3845.99
  152.16  154.55  154.55
BR Coef=-1 , 0 , 0 ,, 0 ,,,0.8,-1,,0,
WSPro=,,,, 1 ,,,, 0 ,,,, 0 ,,,,-1 ,-1 ,-1 , 0 , 0 , 0 , 0 , 0
BC Design=,, 0 ,, 0 ,,,,,,
BC Use User HTab Curves=0
BC User HTab FreeFlow(D)= 0

Type RM Length L Ch R = 1 ,80941.05,420.95,140.21,51.45
BEGIN DESCRIPTION:
Downstream Section - KATY-HOCKLEY CUTOFF RD
END DESCRIPTION:
Node Name=AR
XS GIS Cut Line= 6
2983007.3264891113877071.90777132980449.4762898513874911.2647828
 2980464.0031637 13874442.9907852980478.1373217713873987.3683367
2979794.4543059513872710.78788462977982.0153455313871364.7886081
#Sta/Elev= 30
       0  153.64   67.69  154.17  704.64  152.78  899.54  155.19  1159.4  154.19
 1259.35  151.58 1279.34  154.04 1839.05  151.99 2304.37  155.55 2383.78  152.39
 3752.01  151.87 3801.85  149.13  3816.8  144.85 3866.35  151.56 4287.62  152.73
 4317.58  149.95 4352.53  153.41 4382.49  153.28 4412.46  149.57 4432.43  152.83
 4472.38  153.29 4517.32  149.32 4602.21  153.77 4801.95  154.47 4876.86  152.42
 5141.52  154.14 5236.39  151.69 5555.98   154.2 6235.22  152.64 7978.34  154.16
#Mann= 5 ,-1 , 0
       0     .07       0   67.69     .12       0 2304.37     .07       0
 3752.01     .06       0 3866.35     .07       0
#XS Ineff= 4 ,-1
       0 2283.83  154.56 2283.83  3784.1   151.7 3843.79 6869.54   151.7
 6869.54 7978.34  154.56
Permanent Ineff=
       F       F       F       F
Bank Sta=3752.01,3866.35
XS Rating Curve= 0 ,0
Exp/Cntr=0.5,0.3

Type RM Length L Ch R = 1 ,80800.84,778.24,893.9,612.41
BEGIN DESCRIPTION:
CONFLUENCE WITH U101-12-00
END DESCRIPTION:
XS GIS Cut Line= 6
2982936.5431661213876722.52723642982465.5841342813876234.0613499
2980647.8200532813874507.30988212980527.9098600313874271.1699344
2980529.23006736 13873996.2200252978756.9481788613870650.2181869
#Sta/Elev= 30
       0  153.48  603.69  153.26  618.66  151.11   643.6  153.59  818.37  155.64
  903.28  152.65 1202.94  152.05 1252.88  154.49 1437.67   152.2 1532.56  152.76
 1577.51  155.97 1611.33  152.66 3305.65  152.97 3347.84  144.64  3375.6  152.61
 3400.59  153.42 3870.37  150.62  3945.3  152.83 3965.28  149.68 3990.26  153.25
 4040.21  153.36 4080.17  149.78  4160.1  153.85 4289.98   154.2 4594.69  154.06
  4694.6  151.65  5009.3  153.87 6502.89  154.21 6517.88  152.28 7511.94  154.06
#Mann= 4 ,-1 , 0
       0     .12       0 1611.33     .07       0 3305.65     .06       0
 3400.59     .07       0
#XS Ineff= 2 ,-1
       0  818.37  154.21 6502.89 7511.94  154.21
Permanent Ineff=
       F       F
Bank Sta=3305.65,3400.59
XS Rating Curve= 0 ,0
Exp/Cntr=0.3,0.1

Type RM Length L Ch R = 1 ,79906.94,595.78,751.72,868.13
Node Name=AQ
XS GIS Cut Line= 5
2982948.53198728 13876514.7189252982304.8603743613875632.6002824
2981565.6000418713874310.28009242981185.2799363613873870.7901578
2978885.1739722813870531.9805624
#Sta/Elev= 30
       0  153.65    34.9  151.58  204.44  153.22   219.4  151.34  269.26  153.36
  284.22  151.15  329.09  152.45  349.04  155.06  443.78  152.16 1101.99  153.49
 1131.88  151.51 2496.93  151.91 2701.31  150.18 2726.15  152.34 2760.92  149.82
 2885.11  151.71 2895.05  151.48 2921.53  143.28 2939.76  149.74 2959.63  151.83
 4402.95  150.93 4427.95  152.94 4452.94  152.81 4477.94  149.88 4502.93  153.52
 6002.69  153.57 6012.69  151.65 6042.69  153.62 6197.66  152.01 7242.49  154.17
#Mann= 4 ,-1 , 0
       0     .12       0 1131.88     .07       0 2885.11     .06       0
 2959.63     .07       0
#XS Ineff= 2 ,-1
       0  349.04  153.65 4502.93 7242.49  153.52
Permanent Ineff=
       F       F
Bank Sta=2885.11,2959.63
XS Rating Curve= 0 ,0
Exp/Cntr=0.3,0.1

Type RM Length L Ch R = 1 ,79155.22,832.1,971.66,1033.52
XS GIS Cut Line= 5
2982957.7347247813876319.05921142981959.4699890313873716.0998504
2981941.6301296913873598.54988862981840.4324974413873310.5980367
2979453.2781510213870008.1279356
#Sta/Elev= 30
       0  154.16   54.96   151.7  199.84  151.57  239.81  153.12  319.75   152.1
   384.7  154.68  544.57  154.57  574.55   152.2  699.45  153.13  767.23  151.33
 2218.26  151.62 2243.24  149.09 2253.24  151.58 2802.69  150.39 2817.55  149.98
 2851.82  142.41 2856.61  146.82 2868.68   150.9 2901.77  154.88 2921.49  154.58
  2946.1   150.7  5341.9  152.39  5416.9  150.73  5461.9  152.64  5496.9  149.72
  5511.9  151.85  5726.9   152.4 5881.89  150.88 6791.88  151.24 7286.88  153.02
#Mann= 4 ,-1 , 0
       0     .12       0  767.23     .07       0 2802.69     .05       0
 2868.68     .07       0
#XS Ineff= 2 ,-1
       0  699.45  152.64  5461.9 7286.88  152.64
Permanent Ineff=
       F       F
Bank Sta=2802.69,2868.68
XS Rating Curve= 0 ,0
Exp/Cntr=0.3,0.1

Type RM Length L Ch R = 1 ,78183.56,880.48,976.46,807.05
Node Name=AP
XS GIS Cut Line= 5
2983285.3754113513875073.1736412  2982830.159849  13873703.13006
  2982812.319989 13873598.549889  2982648.099845 13872735.969921
  2980125.296164 13869388.455947
#Sta/Elev= 30
 1383.74  151.41 2148.05  150.13 2227.98  151.83 2856.46  149.38 2881.29  140.42
 2885.02  141.83  2886.8  145.09 2895.28  145.67  2904.5  150.05 2933.52  153.48
 2963.46  150.14 3033.31  149.48 4171.33  151.46 5195.53  149.27 5904.98  150.63
 5974.92  152.96 6014.89  158.61 6064.85   152.4 6119.81  152.47 6159.78  159.45
 6179.76  157.71 6204.74  151.72  6254.7  151.21 7178.98  151.61 7208.96  149.48
 7258.92  151.82  7288.9  149.65 7303.88   152.8 7453.77  150.95 8003.34  152.31
#Mann= 3 ,-1 , 0
 1383.74     .07       0 2856.46     .05       0  2904.5     .07       0
#XS Ineff= 3 ,-1
 1383.74 1638.51  152.09 6159.78 7303.88  151.45 7303.88 8003.34   152.8
Permanent Ineff=
       F       F       F
Bank Sta=2856.46,2904.5
XS Rating Curve= 0 ,0
Exp/Cntr=0.3,0.1

Type RM Length L Ch R = 1 ,77207.09,975.6,1123.62,840.07
Node Name=AO
XS GIS Cut Line= 6
2983969.8334513613875138.98073892983882.7194233513874383.9981209
2983700.85003644 13873558.0201142983670.0400586913873424.2500404
2983137.67235702 13872288.046276 2980361.1841436 13869170.942274
#Sta/Elev= 30
  894.98  150.76 1464.97  151.58 1559.97  149.67 1629.97  151.64 1669.89  151.59
 1694.77  149.53 1724.62  151.27 1819.14  149.28 2535.05  149.17 2563.47  144.37
 2577.77  143.74 2583.69  139.66 2586.88  139.93 2600.55  148.66  2613.5  149.82
 3747.78  148.81 3947.74  150.73 4047.72  149.07 4637.63  148.98 6567.33  151.34
 6597.33  149.98 7177.23  152.71 7642.16  151.52 7667.16  149.32 7692.15  151.89
 7717.15  151.76 7737.15  149.13 7757.14  153.13 7787.14  151.84  8067.1  151.73
#Mann= 3 ,-1 , 0
  894.98     .07       0 2535.05     .05       0  2613.5     .07       0
#XS Ineff= 2 ,-1
  894.98 1464.97  151.58 7177.23  8067.1  151.58
Permanent Ineff=
       F       F
Bank Sta=2535.05,2613.5
XS Rating Curve= 0 ,0
Exp/Cntr=0.3,0.1

Type RM Length L Ch R = 1 ,76083.47,908.54,904.88,743.77
XS GIS Cut Line= 6
2984703.2348426913875383.70215822984791.2290892813874353.6284309
2984496.1499550313873046.4601135 2984389.939865613872930.5298992
2983536.0452479413871669.14003352980621.7512077813868930.6717572
#Sta/Elev= 30
       0  151.05  928.95  151.44 1008.85  148.84 1043.79  150.78 1382.54  149.33
  1502.1  150.67  2368.9  147.71 2413.19  149.22 2427.93  147.76 2439.14  142.12
 2442.12  138.77 2445.39  138.45 2453.74  143.22 2470.81  143.68  2491.8  147.33
 2715.89  147.55 2890.69  145.27 3005.55   145.5 3120.42  148.55 4094.31  149.95
 5893.87   149.3 6068.83  149.59 6098.82   151.2 6348.76  149.17 6388.75     151
 6433.74  149.39 7988.36  151.71 8013.35  148.44 8028.35  151.77 8053.34  152.28
#Mann= 3 , 0 , 0
       0     .07       0 2427.93     .05       0  2491.8     .07       0
#XS Ineff= 2 ,-1
       0 1043.29   150.2 6098.82 8053.34   150.2
Permanent Ineff=
       F       F
Bank Sta=2427.93,2491.8
XS Rating Curve= 0 ,0
Exp/Cntr=0.3,0.1

Type RM Length L Ch R = 1 ,75178.59,422.56,1164.83,1023.23
XS GIS Cut Line= 6
2985627.8707886913874439.21224932985647.9327564413873592.7487191
2985137.4101554513872545.44996072985001.20996852 13872508.160009
2983743.2594004413870887.15275242981558.6935596213868963.6684103
#Sta/Elev= 30
       0  149.77   32.78  148.64   61.16  150.27  170.54  149.72  200.37  151.04
  503.65  149.22  627.94  150.81  747.27  149.25   777.1  150.73 1230.09  148.86
 1314.73  150.12 1508.92   147.7  2060.5   148.1 2070.24  146.56 2088.01  139.11
  2092.3  138.88 2097.72  142.73  2109.2  142.84    2119   146.6 2128.67  147.16
 2362.69  147.15 2417.61  144.81 2497.49  147.13 3101.56  149.58 3151.48     148
 3895.34  149.78 4579.32  148.36 7045.71  151.16 7080.66  148.44 7115.61     151
#Mann= 3 , 0 , 0
       0     .07       0  2060.5     .06       0 2128.67     .07       0
#XS Ineff= 2 ,-1
       0 1314.73   149.5 5013.68 7115.61   149.5
Permanent Ineff=
       F       F
#Block Obstruct= 2 , 0
       0   61.16  150.27               0
Bank Sta=2060.5,2128.67
XS Rating Curve= 0 ,0
Exp/Cntr=0.3,0.1

Type RM Length L Ch R = 1 ,74013.76,35.62,30.21,205.05
Node Name=AN
XS GIS Cut Line= 6
2985695.5617576813873396.93546142985719.0198846213872573.6900617
2985740.1500916913872131.27985732985739.8298823513872033.5799214
2985218.8299401113870901.88008512984225.91525927 13869052.741723
#Sta/Elev= 30
 1043.59  148.64 1223.28  147.54 1298.15  148.18 1392.99  147.07  1442.9  147.61
 1467.86  146.82 1662.52  146.82 1782.32  148.11 1817.26   147.1 2220.88  146.95
 2290.26  145.81 2314.97  146.75 2349.16  143.02 2366.87   139.7 2368.46  138.65
 2412.82  142.76 2427.72  145.28 2452.63  143.45 2507.45  146.31 2701.81  146.39
 2796.49  147.84 4148.39  148.01 4213.35   148.9 4248.33   148.1 4478.21  147.76
 5662.55  148.43 5697.53  149.13 5712.53  146.39 5732.51  148.58  5752.5  149.09
#Mann= 3 ,-1 , 0
 1043.59     .07       0 2314.97     .06       0 2427.72     .07       0
#XS Ineff= 3 ,-1
 1043.59 2242.31  146.36 2447.16 3155.31  146.09 4213.35  5752.5   148.9
Permanent Ineff=
       F       F       F
Bank Sta=2314.97,2427.72
XS Rating Curve= 0 ,0
Exp/Cntr=0.5,0.3
